--- BvrCrk.prj (project) ---

Proj Title=BvrCrk
Current Plan=p01
Default Exp/Contr=0,0
English Units
Geom File=g01
Flow File=f01
Plan File=p01
BEGIN DESCRIPTION:
END DESCRIPTION:
DSS Export Rating Curves= 0
DSS Export Rating Curve Sorted= 0
DSS Export Volume Flow Curves= 0
DXF OffsetX= 0
DXF OffsetY= 0
DXF ScaleX= 0
DXF ScaleY= 0

--- BvrCrk.p01 (plan) ---

Plan Title=Floodplain
Program Version=4.00
Geom File=g01
Flow File=f01
K Sum by GR=0
Std Step Tol=0.01
Critical Tol=0.01
Num of Std Step Trials=20
Max Error Tol=0.3
Flow Tol Ratio=0.001
Split Flow NTrial=30
Split Flow Tol=0.02
Split Flow Ratio=0.02
Log Output Level=0
Friction Slope Method=1
Unsteady Friction Slope Method=2
Unsteady Bridges Friction Slope Method=1
Global Log Level=0
CheckData=False
Run HTab=0
Run UNet=0
Run PostProcess=0
UNET Theta=0
UNET Theta Warmup=0
UNET ZTol=0
UNET ZSATol=0
UNET MxIter=0
UNET MaxInSteps=0
UNET DtIC=0
UNET DtMin=0
UNET MaxCRTS=0
UNET WFStab=0
UNET SFStab=0
UNET WFX=0
UNET SFX=0
UNET DSS MLevel=0
UNET DZMax Abort=0
UNET Convert EG Bridges=0
UNET Use Existing IB Tables=0
UNET Froude Limit=0
UNET Froude Power=0
Write IC File=0
Echo Input=False
Echo Output=False
Write Detailed=0

--- BvrCrk.f01 (steady flow) ---

Flow Title=NFF Regression Equation
Program Version=4.10
Number of Profiles= 1
Profile Names=P100yr
River Rch & RM=BvrCrk,Main            ,28866.2
375.3533
River Rch & RM=BvrCrk,Main            ,28336.4
596.3137
River Rch & RM=BvrCrk,Main            ,25735.2
661.3199
River Rch & RM=BvrCrk,Main            ,25214.9
728.5631
River Rch & RM=BvrCrk,Main            ,24046.2
736.1474
River Rch & RM=BvrCrk,Main            ,23539.5
1421.618
River Rch & RM=BvrCrk,Main            ,19890.4
1491.869
River Rch & RM=BvrCrk,Main            ,11790.6
1647.025
River Rch & RM=BvrCrk,Main            ,11505.9
2212.906
River Rch & RM=BvrCrk,Main            ,10840.4
2215.781
River Rch & RM=BvrCrk,Main            ,10157.1
2461.188
River Rch & RM=BvrCrk,Main            ,393.8
2656.738
Boundary for River Rch & Prof#=BvrCrk,Main            , 1
Up Type= 0
Dn Type= 1
Dn Known WS=2290.5
DSS Import GetInterval= 0
DSS Import GetPeak= 0
DSS Import FillOption= 0

--- BvrCrk.g01 (geometry) ---

Geom Title=USGS 3m DEM
Program Version=4.10

River Reach=BvrCrk          ,Main
Reach XY= 30
     1931763.899      242804.904     1932241.876        244653.6
      1933012.01      246106.669     1933560.887      246360.631
     1933719.741      246726.517     1931850.375      248980.937
     1930828.061      251522.885     1930958.264      252217.508
     1930770.522      253007.767     1927870.662      254795.498
     1927114.012      255663.227      1926043.77      255742.824
     1925922.413      256095.638     1926023.126      256925.736
     1925810.886      256949.173     1925439.047      256536.229
     1924933.282      256899.694     1924704.116       257584.59
      1924706.72      258755.163     1925021.824       258872.35
     1925042.083      259451.262     1925343.439      259496.048
      1925088.23      259675.736     1925530.556      260273.694
     1924667.903      261072.047     1924439.811      261058.123
      1924646.78      261503.647     1924970.986      261547.154
     1925094.057       262085.38     1925436.325      262206.017

Type RM Length L Ch R = 1 ,28866.2 ,529.5,529.9,530.3
XS GIS Cut Line= 3
     1931377.347      242937.166     1931766.977      242811.154
     1932156.607      242685.143
#Sta/Elev= 30
       0  2633.3    49.9 2633.26    89.9 2633.82   129.8 2633.47   149.8 2632.61
   169.8 2630.94   189.8 2629.97   229.7    2629   289.6 2626.45   319.6 2624.34
   339.6 2622.24   369.6 2620.48   399.5  2620.2     401  2620.2     416  2620.2
   449.4  2620.2   479.4 2620.82   569.3 2621.28   579.3 2622.06   589.3 2623.52
   659.2 2628.64   669.2 2629.99   679.2  2630.6   699.2 2630.94   719.1 2630.27
   729.1 2630.31   739.1 2630.54   759.1 2631.72     799 2633.02     819 2633.37
#Mann= 3 , 0 , 0
       0     .06       0     401    .045       0     416     .06       0
Bank Sta=401,416
XS Rating Curve= 0 ,0
Exp/Cntr=0.3,0.1

Type RM Length L Ch R = 1 ,28336.4 ,165.3,168.1,170.9
XS GIS Cut Line= 3
     1931068.216      243404.225     1931667.705      243389.343
     1932327.534      243193.593
#Sta/Elev= 30
       0 2648.02      60  2648.2   109.9 2649.46   199.9    2651   219.9  2650.6
   289.8 2648.05   309.8 2647.01   349.8  2645.9   389.8 2645.52   479.7 2645.74
   529.7 2645.08   579.7 2645.58   599.7 2645.44   649.6 2644.25   709.4  2643.9
   719.4 2642.87   729.3 2640.96   789.2 2626.61   809.1 2620.76   829.1  2620.2
   858.2  2620.2   873.2  2620.2   958.8 2620.28  1018.6 2625.12  1058.5 2627.81
  1128.3 2631.52  1138.3 2632.56  1208.1 2636.08  1228.1 2637.44  1287.9 2639.69
#Mann= 3 , 0 , 0
       0     .06       0   858.2    .045       0   873.2     .06       0
Bank Sta=858.2,873.2
XS Rating Curve= 0 ,0
Exp/Cntr=0.3,0.1

Type RM Length L Ch R = 1 ,28168.2 ,191.2,180.7,170.2
XS GIS Cut Line= 3
     1930981.381      243461.383     1931781.684      243498.566
     1932578.446      243379.937
#Sta/Elev= 30
       0 2648.72    98.9 2645.17   158.3 2643.88   217.6 2644.63   356.1 2649.07
   494.6 2648.34   563.8 2648.77     633 2647.79   712.2 2642.34   781.4 2634.69
   791.3  2633.4   811.1 2627.49     831 2623.33   850.9 2620.77   870.8 2620.19
   890.7 2621.21   933.8  2620.2   948.8  2620.2    1020 2620.46    1199  2630.6
  1278.5 2637.09  1298.4 2639.44  1358.1 2643.21    1368  2644.4  1387.9 2648.22
  1447.6 2654.77  1467.5 2657.81  1527.2 2663.18    1547 2665.93  1606.7 2671.43
#Mann= 3 , 0 , 0
       0     .06       0   933.8    .045       0   948.8     .06       0
Bank Sta=933.8,948.8
XS Rating Curve= 0 ,0
Exp/Cntr=0.3,0.1

Type RM Length L Ch R = 1 ,27987.5 ,183.9,188.9,193.8
XS GIS Cut Line= 5
     1931123.028      243941.211     1931563.246      243935.278
     1931726.796      243762.382     1932165.901      243514.501
     1932574.905      243452.531
#Sta/Elev= 30
       0 2664.91      20 2660.82      70 2653.93   180.1 2650.53   250.2 2643.39
   270.2 2640.14   310.2 2636.09   330.2 2636.44   370.2 2638.91   440.3 2644.33
   489.8 2642.06   529.5 2645.53   559.3 2644.83   579.1  2642.8   608.8 2637.29
   648.5 2634.97   767.2 2621.66   816.7  2620.2   886.9  2620.2   901.9  2620.2
   984.8 2620.54  1034.2 2623.65  1152.8 2628.18  1202.2 2630.91    1281 2632.27
  1320.4 2634.52  1359.8 2638.45  1389.3 2645.64  1468.1  2659.3  1596.2 2671.95
#Mann= 3 , 0 , 0
       0     .06       0   886.9    .045       0   901.9     .06       0
Bank Sta=886.9,901.9
XS Rating Curve= 0 ,0
Exp/Cntr=0.3,0.1

Type RM Length L Ch R = 1 ,27798.7 ,263.6,263,262.4
XS GIS Cut Line= 2
     1931478.915      244035.052     1932484.681      243616.695
#Sta/Elev= 30
       0 2641.24      60 2646.12      70 2648.44    89.9 2650.43   179.9 2655.31
   219.9 2659.51   229.8 2659.26   249.8 2654.38   259.8 2653.61   299.8 2653.84
   319.8 2652.38   379.8  2641.6   399.8 2635.59   409.7 2631.78   419.7  2626.5
   439.7 2621.07     522 2612.84   529.7 2612.32     537 2612.44   589.6 2616.42
   609.6 2619.38   679.6 2626.78   689.6 2628.75   749.5 2633.06   789.5 2634.76
   879.4 2633.86   929.4 2635.41  1019.4  2646.8  1039.3 2650.84  1089.3 2658.52
#Mann= 3 , 0 , 0
       0     .06       0     522    .045       0     537     .06       0
Bank Sta=522,537
XS Rating Curve= 0 ,0
Exp/Cntr=0.3,0.1

Type RM Length L Ch R = 1 ,27535.6 ,273.1,279.8,284.8
XS GIS Cut Line= 3
     1931722.275      244229.831     1932095.903      244062.225
     1932469.531      243894.618
#Sta/Elev= 30
       0 2665.26    69.9 2663.79    99.9 2662.13   109.9 2660.86   149.8 2654.24
   159.8 2651.16   169.8 2646.47   239.7 2626.59   249.7 2622.53   259.7 2619.21
   269.7 2618.29   329.6 2614.96   349.6 2613.02   371.1 2611.61   379.5 2611.47
   386.1 2611.89   419.5 2614.49   449.4 2617.78   499.4  2622.3   509.4 2623.34
   519.4 2625.09   589.3 2631.67   609.3 2634.64   679.2 2641.26   699.2 2644.29
   719.1 2646.33   769.1 2650.88     779 2652.21     809 2654.63     819 2655.07
#Mann= 3 , 0 , 0
       0     .06       0   371.1    .045       0   386.1     .06       0
Bank Sta=371.1,386.1
XS Rating Curve= 0 ,0
Exp/Cntr=0.3,0.1

Type RM Length L Ch R = 1 ,27255.8 ,409.5,400.4,392.2
XS GIS Cut Line= 3
     1931738.231      244383.682     1932144.154      244331.419
      1932546.76      244249.848
#Sta/Elev= 30
       0  2658.3    39.9 2656.44    59.9 2654.06   119.8 2649.32   159.7 2644.67
   169.7 2642.66   199.6 2633.93   209.6 2630.54   219.6 2624.68   229.6 2621.96
   239.6  2620.1   289.5 2616.99   369.3 2611.17   389.3 2608.42   401.4 2607.47
   409.3 2607.26   416.4  2607.5   428.8 2608.55     468 2613.85   536.4 2619.27
     556 2621.51   624.4 2627.13   634.2  2629.2   692.9  2636.8   702.7 2638.53
   722.2 2643.94   751.6 2648.87   790.7 2654.53   800.5 2656.93   820.1 2659.44
#Mann= 3 , 0 , 0
       0      .1       0   401.4    .045       0   416.4      .1       0
Bank Sta=401.4,416.4
XS Rating Curve= 0 ,0
Exp/Cntr=0.3,0.1

Type RM Length L Ch R = 1 ,26855.4 ,426.6,432.5,439.2
XS GIS Cut Line= 3
     1931921.204      244913.094     1932274.679      244706.446
     1932621.145      244487.605
#Sta/Elev= 30
       0  2638.1    59.9 2637.18   159.8 2637.84   169.8 2637.69   179.8 2636.92
   189.7 2635.71   219.7 2630.68   229.7 2628.08   239.7 2624.96   259.6 2620.42
   289.6 2614.15   299.6 2612.61   329.6 2609.73   369.5 2607.71   400.3 2605.68
   409.4 2605.44   415.3 2605.88   439.4 2608.46   449.4 2609.27   529.4 2614.82
   559.4 2618.02   599.4 2623.16   659.3 2637.15   679.3 2640.09   689.3 2641.23
   699.3    2642   729.3 2646.16   789.3 2656.07   799.2 2658.45   819.2 2661.83
#Mann= 3 , 0 , 0
       0      .1       0   400.3    .045       0   415.3      .1       0
Bank Sta=400.3,415.3
XS Rating Curve= 0 ,0
Exp/Cntr=0.3,0.1

Type RM Length L Ch R = 1 ,26422.8 ,363.4,362.3,360.5
XS GIS Cut Line= 2
     1932102.795      245167.671     1932899.379       244931.46
#Sta/Elev= 30
       0 2653.56    29.7 2653.36    79.1 2652.06    98.9 2650.95   138.5 2647.66
   158.3 2644.95   187.9 2640.17   197.8 2637.52   237.4 2629.89   257.2 2625.68
   267.1 2623.29     277 2620.29   286.8 2616.68   306.6 2612.63   336.3 2607.19
   346.2 2605.79     366  2604.5   407.8 2602.77   415.4 2602.64   422.8 2602.78
   464.9 2605.64   563.8 2608.83   603.4 2611.25   642.9  2615.6   692.4 2622.37
   702.3 2624.41   751.7 2631.45   771.5 2633.36   791.3 2636.19   830.9 2640.03
#Mann= 3 , 0 , 0
       0      .1       0   407.8    .045       0   422.8      .1       0
Bank Sta=407.8,422.8
XS Rating Curve= 0 ,0
Exp/Cntr=0.3,0.1

Type RM Length L Ch R = 1 ,26060.4 ,216,215,214.9
XS GIS Cut Line= 3
     1932271.322      245500.572     1932662.268      245366.059
     1933043.491      245218.444
#Sta/Elev= 30
       0 2652.64    29.5 2654.84    59.1 2655.04    98.4 2653.47     128 2650.15
   147.7 2646.63   167.3 2640.15   177.2 2636.42     187 2631.68   196.9    2625
   246.1  2605.1   255.9 2602.15   275.6 2600.25   403.6  2596.9   404.8 2596.93
   419.8 2597.49   453.3 2599.38   523.1 2601.39   543.1 2602.78   612.9 2618.36
   622.8 2621.21   632.8 2625.64   702.6 2646.36   722.5 2655.28   742.5 2660.03
   762.4  2662.5   772.4 2662.67   792.3 2662.41   802.3 2660.88   822.2 2659.81
#Mann= 3 , 0 , 0
       0      .1       0   404.8    .045       0   419.8      .1       0
Bank Sta=404.8,419.8
XS Rating Curve= 0 ,0
Exp/Cntr=0.3,0.1

Type RM Length L Ch R = 1 ,25845.3 ,113.1,110.1,107.1
XS GIS Cut Line= 2
     1932413.858      245688.276     1933162.814      245401.441
#Sta/Elev= 30
       0 2636.18    29.7 2629.08    49.5 2621.19   118.8 2604.56   138.6 2600.67
   148.5 2599.78   217.8 2595.94   227.7 2595.04   344.7 2590.95   359.7 2590.51
   366.4  2590.5     406 2593.12   465.4 2596.18     505 2598.72   534.7 2601.54
   544.6 2602.76   554.5 2604.36   564.4 2608.19   574.3 2612.58   584.2 2615.47
   594.1    2618   613.9 2622.28   643.6 2627.55   653.5 2631.65   663.4 2634.63
     703 2644.86   742.6 2653.39   772.3 2655.94   782.2 2657.31     802 2661.08
#Mann= 3 , 0 , 0
       0      .1       0   344.7    .045       0   359.7      .1       0
Bank Sta=344.7,359.7
XS Rating Curve= 0 ,0
Exp/Cntr=0.3,0.1

Type RM Length L Ch R = 1 ,25735.2 ,529.5,520.2,510.8
XS GIS Cut Line= 3
     1932026.101      246017.604     1932475.828      245831.693
     1933158.947      245460.646
#Sta/Elev= 30
       0 2620.06    29.8 2616.96    79.4 2614.46    99.3 2616.31   158.9 2627.06
   258.2 2640.71   297.9 2642.72   377.4 2641.63     427 2633.38   446.9 2628.76
   466.8 2621.82   476.7 2614.89   486.6 2611.47   526.5 2600.24   546.4 2596.81
   566.4 2595.29   825.5  2587.8   841.7 2586.59   845.4 2586.34   856.7 2586.49
  1004.9 2597.19  1014.9 2599.32  1024.8 2602.96  1094.6 2622.59  1104.6 2626.44
  1114.5 2631.75  1194.3  2655.7  1204.2  2660.8  1224.2 2664.21    1264 2666.27
#Mann= 3 , 0 , 0
       0      .1       0   841.7    .045       0   856.7      .1       0
Bank Sta=841.7,856.7
XS Rating Curve= 0 ,0
Exp/Cntr=0.3,0.1

Type RM Length L Ch R = 1 ,25214.9 ,298.9,298.6,297.4
XS GIS Cut Line= 3
     1932651.116      246601.896     1932863.586      246297.356
     1933359.349      245667.029
#Sta/Elev= 30
       0 2649.66   117.3 2643.93   185.7 2638.79   205.2 2631.74   234.5 2624.35
   254.1 2616.86   312.7 2601.19   332.2 2598.24   391.1 2584.69   410.9 2583.28
   440.6 2583.55   460.4 2581.59   470.3 2578.64   480.2 2572.42   490.1 2568.35
     500  2567.4   605.6  2567.4   620.6  2567.4   737.6 2567.39   757.4 2569.61
   787.2 2575.61     807 2577.36   846.6 2586.02     906 2601.56   915.8  2602.4
   945.6 2611.36  1034.7 2643.55  1044.6  2644.9  1123.8 2669.46  1173.3 2680.17
#Mann= 3 , 0 , 0
       0      .1       0   605.6    .045       0   620.6      .1       0
Bank Sta=605.6,620.6
XS Rating Curve= 0 ,0
Exp/Cntr=0.3,0.1

Type RM Length L Ch R = 1 ,24916.1 ,539.5,541.9,541.7
XS GIS Cut Line= 2
     1932981.841      246630.241     1933446.753      245898.375
#Sta/Elev= 30
       0  2649.1    49.8 2646.89    59.8    2646    69.8 2643.74    79.7 2640.56
    99.7 2631.55   109.6 2627.94   119.6 2624.75   129.6 2623.47   199.3  2599.9
   219.2 2593.44   239.2 2589.14   249.2  2585.3     299 2570.48     309 2567.94
   318.9 2567.38   401.1  2567.4   416.1  2567.4   617.9 2567.51   627.9 2568.76
   657.8 2574.53   667.7 2576.04   677.7 2576.65   697.6 2581.46   737.5 2589.56
   777.4 2599.53   787.3 2601.09   797.3 2602.11   827.2 2610.38     867 2623.28
#Mann= 3 , 0 , 0
       0      .1       0   401.1    .045       0   416.1      .1       0
Bank Sta=401.1,416.1
XS Rating Curve= 0 ,0
Exp/Cntr=0.3,0.1

Type RM Length L Ch R = 1 ,24373.9 ,302.8,327.7,355.2
XS GIS Cut Line= 3
     1933265.958      246737.555     1933516.088      246566.416
     1934051.979       245911.59
#Sta/Elev= 30
       0 2603.09     9.8 2601.28    29.3 2594.79    48.9 2591.59    97.8 2575.95
   107.5 2574.06   283.5 2570.75   303.1 2570.14     323 2567.44   332.9  2567.4
   353.8  2567.4   368.8  2567.4   402.6 2567.78   422.5 2571.15   432.5 2571.85
   502.2 2568.48   551.9 2568.55   671.4 2575.43   701.3 2580.27   711.2 2580.16
   810.8 2597.43   830.7 2599.21   840.6 2598.43   940.2 2612.18   960.1 2611.18
  1019.8 2621.98  1039.7 2624.72  1059.6 2626.16  1079.5 2622.84  1149.2 2624.62
#Mann= 3 , 0 , 0
       0      .1       0   353.8    .045       0   368.8      .1       0
#XS Ineff= 2 , 0
                          441.53         2571.69
Permanent Ineff=
       F       F
Bank Sta=353.8,368.8
XS Rating Curve= 0 ,0
Exp/Cntr=0.3,0.1

Type RM Length L Ch R = 1 ,24046.2 ,78.2,81.7,85.2
XS GIS Cut Line= 3
     1933378.825       246704.59     1933943.381      246812.206
     1934441.175      246269.027
#Sta/Elev= 30
       0 2574.09    79.3 2574.07   128.8 2577.06   138.7 2575.91   158.5 2569.05
   178.4 2565.19     218 2561.85   287.4  2560.6   297.3 2558.98   317.1 2551.62
   325.6 2550.86     327 2550.73   340.6 2552.22   406.3 2564.63   455.8 2571.17
   554.9 2575.81   604.6 2584.91   664.3 2586.83   704.2 2591.65   753.9 2594.65
   823.6 2594.19   843.6 2595.78   903.3 2593.55   943.1 2593.95     963 2595.97
  1032.7 2590.02  1082.5 2593.04  1152.2 2588.69    1202 2591.28  1311.5 2592.18
#Mann= 3 , 0 , 0
       0      .1       0   325.6    .045       0   340.6      .1       0
Bank Sta=325.6,340.6
XS Rating Curve= 0 ,0
Exp/Cntr=0.3,0.1

Type RM Length L Ch R = 1 ,23964.5 ,420,424.7,430.3
XS GIS Cut Line= 6
     1933320.396      246780.725     1933630.248       246826.76
     1933709.924      246855.089     1933761.271      246869.254
     1934009.153      246855.089     1934271.199      246892.272
#Sta/Elev= 30
       0 2584.54    29.4 2576.72    39.2 2574.84      49 2574.02    68.5 2574.72
   117.5 2578.19   195.8  2570.9   205.6 2569.13   225.2 2567.09   293.7 2563.92
   313.2 2560.97   350.8 2551.64   357.9 2550.95   360.2 2550.73   369.6  2551.4
   372.9 2552.54   388.4 2557.94   397.8  2559.8   451.1 2568.64   470.9 2570.94
     610 2573.87   659.6 2576.33   709.2 2582.19   777.8 2586.69   797.4 2590.22
   826.8    2597   856.2 2600.42     866 2600.86   934.6 2598.47     964 2599.64
#Mann= 3 , 0 , 0
       0      .1       0   357.9    .045       0   372.9      .1       0
Bank Sta=357.9,372.9
XS Rating Curve= 0 ,0
Exp/Cntr=0.3,0.1

Type RM Length L Ch R = 1 ,23539.5 ,272.7,279.3,285.9
XS GIS Cut Line= 2
     1933053.797      246931.798     1934065.811      247584.569
#Sta/Elev= 30
       0 2621.59    49.8 2612.55    69.7 2606.83    89.6 2596.22   109.5 2587.36
   139.3 2577.34   149.3 2575.98     199 2579.94     209 2579.82   278.7 2572.94
   318.5  2570.9   358.3 2563.55   378.2 2557.88   408.1 2551.25     418 2550.56
   428.7 2551.28   443.7 2553.78   527.5 2566.64   557.4 2566.04   567.3 2565.18
   587.2 2561.44   607.1 2560.89   766.4  2578.7   955.5 2584.88   975.4 2587.22
   995.3 2588.18    1045 2596.05  1074.9 2599.28  1174.4 2616.56  1204.3 2619.02
#Mann= 3 , 0 , 0
       0      .1       0   428.7    .045       0   443.7      .1       0
Bank Sta=428.7,443.7
XS Rating Curve= 0 ,0
Exp/Cntr=0.3,0.1

Type RM Length L Ch R = 1 ,23260.2 ,294,290,286
XS GIS Cut Line= 2
     1932954.945      247047.323     1933488.601      247673.098
#Sta/Elev= 30
       0 2594.85    29.7 2590.17    79.3 2585.04   128.8 2577.29   158.5 2579.78
   178.4 2579.99   198.2 2581.89   208.1 2582.04   227.9 2580.18   277.4 2573.74
   317.1 2569.57   366.6  2558.4   386.4 2551.08   396.4 2550.52     407 2550.72
     422 2551.53   505.4 2561.54   525.2  2564.6   554.9 2566.92   574.7  2567.2
   604.4 2564.42   614.3 2564.37   624.2 2565.78     654 2576.76   673.8 2581.38
   693.6 2583.77   753.1 2595.34   792.7 2604.21   802.6 2605.05   822.4 2608.64
#Mann= 3 , 0 , 0
       0      .1       0     407    .045       0     422      .1       0
Bank Sta=407,422
XS Rating Curve= 0 ,0
Exp/Cntr=0.3,0.1

Type RM Length L Ch R = 1 ,22970.1 ,397.3,399.2,400.2
XS GIS Cut Line= 3
     1932707.344        247310.8     1933025.013       247571.38
     1933341.222      247830.886
#Sta/Elev= 30
       0 2654.52     9.8 2654.46    19.6 2650.71    58.7 2629.65    78.3 2623.37
   107.6 2607.42   117.4 2601.38   127.2 2593.54     137  2588.4   146.7 2584.95
   176.1 2583.63   205.4 2584.86   273.9  2579.9   283.7    2578     313 2568.97
   322.8 2565.12   332.6 2557.54   342.4 2552.28   352.2 2550.05     362 2549.81
   371.7  2550.4   580.5 2568.76   610.4 2569.24   630.4 2565.73   640.4 2566.31
   670.3 2580.21   700.2 2589.42   730.1 2601.94   740.1 2604.97   819.9 2615.48
#Mann= 3 , 0 , 0
       0      .1       0   352.2    .045       0   371.7      .1       0
Bank Sta=352.2,371.7
XS Rating Curve= 0 ,0
Exp/Cntr=0.3,0.1

Type RM Length L Ch R = 1 ,22570.7 ,398.7,400,402.1
XS GIS Cut Line= 3
     1932433.169      247578.966     1932761.406      247846.306
     1933091.594      248099.627
#Sta/Elev= 30
       0  2642.6    49.2 2626.76    59.1  2622.8    68.9 2617.81    88.6 2611.34
    98.4 2608.14   118.1 2604.06   157.5 2591.73   167.4 2587.64   177.2 2585.68
   206.7 2585.84   236.3 2587.12   246.1 2585.67   354.4  2557.1   364.3 2553.89
   374.1 2549.16     384 2547.82   403.6 2548.51   522.4 2555.97   581.9 2561.34
   631.4  2571.4   651.2 2574.01   661.1 2574.18     671 2573.24   690.9 2565.83
   700.8 2565.82   730.5 2570.83     780 2581.04   799.9 2586.07   839.5 2592.42
#Mann= 3 , 0 , 0
       0      .1       0     384    .045       0   403.6      .1       0
Bank Sta=384,403.6
XS Rating Curve= 0 ,0
Exp/Cntr=0.3,0.1

Type RM Length L Ch R = 1 ,22170.5 ,404.4,399.6,394.7
XS GIS Cut Line= 3
     1932164.437      247814.986     1932461.926      248096.394
     1932759.415      248377.803
#Sta/Elev= 30
       0 2653.43    69.9 2648.03    89.9 2645.42    99.9 2642.79   119.8 2631.69
   149.8 2616.87   169.8 2611.17   219.7 2586.89   229.7 2585.58   269.7 2586.28
   299.6 2583.65   309.6 2579.82   339.6  2565.5   389.5 2547.47   399.5 2544.38
   404.2 2544.08   409.5 2543.75   419.2 2544.06   569.3 2546.74   659.2 2555.24
   669.2 2558.14   699.2 2572.36   709.1 2576.03   719.1 2577.47   759.1 2577.92
   769.1 2576.29     789 2567.67     799 2564.63     809 2563.96     819  2566.7
#Mann= 3 , 0 , 0
       0      .1       0   404.2    .045       0   419.2      .1       0
Bank Sta=404.2,419.2
XS Rating Curve= 0 ,0
Exp/Cntr=0.3,0.1

Type RM Length L Ch R = 1 ,21770.9 ,399.8,400,400.2
XS GIS Cut Line= 3
     1931865.702      248195.244      1932216.39      248406.687
     1932567.077      248618.131
#Sta/Elev= 30
       0 2562.52   119.8 2562.23   149.8 2564.58   179.8 2562.59   189.8  2563.7
   199.8 2566.24   229.7 2580.45   239.7 2581.94   269.7 2580.62   279.7 2579.98
   299.6 2574.43   339.6  2555.5   349.6 2549.58   359.6 2545.96   389.5 2539.42
   403.7 2537.61   409.5 2537.35   418.7 2537.74   449.4 2540.79   519.4  2544.7
   549.3 2548.14   589.3 2551.16   679.2  2560.8   689.2 2562.62   729.1 2576.75
   739.1 2577.79   769.1 2577.66     779 2576.02     809 2568.03     819 2567.88
#Mann= 3 , 0 , 0
       0      .1       0   403.7    .045       0   418.7      .1       0
Bank Sta=403.7,418.7
XS Rating Curve= 0 ,0
Exp/Cntr=0.3,0.1

Type RM Length L Ch R = 1 ,21370.9 ,405.4,399.6,394.3
XS GIS Cut Line= 3
     1931660.114      248533.432     1932008.869      248748.049
     1932357.623      248962.666
#Sta/Elev= 30
       0 2583.15      30 2578.86    69.9 2577.83   109.9 2573.91   119.8 2571.44
   129.8 2569.89   189.8 2570.46   199.8 2572.71   209.7 2575.88   219.7 2577.16
   269.7 2573.14   299.6 2567.57   369.6 2541.08   379.5 2537.95   409.5 2532.18
   419.5 2530.95   429.5 2531.56   489.4 2539.22   589.3 2544.43   619.2 2547.17
   629.2 2548.98   639.2 2552.18   689.2 2570.55   699.2 2573.63   749.1 2570.52
   759.1 2571.88     779 2579.15     789  2584.2     799 2586.99     819  2587.8
#Mann= 3 , 0 , 0
       0      .1       0   409.5    .045       0   429.5      .1       0
Bank Sta=409.5,429.5
XS Rating Curve= 0 ,0
Exp/Cntr=0.3,0.1

Type RM Length L Ch R = 1 ,20971.2 ,396.1,400.2,403.9
XS GIS Cut Line= 3
     1931412.503      248966.701     1931804.049      249086.563
      1932193.15       249214.54
#Sta/Elev= 30
       0 2591.71    99.9  2580.8   129.8 2580.12   139.8 2579.08   199.8  2565.3
   249.7 2565.96   269.7 2564.45   289.6 2560.76   329.6 2555.34   369.5 2543.45
   379.5 2537.75   389.5  2534.6   399.5 2532.21   419.5 2529.38   429.5 2529.03
   439.4 2529.68   469.4 2534.27   589.3 2540.82   599.3 2542.93   619.3 2548.91
   629.3 2553.98   639.3 2557.66   659.2  2563.4   679.2 2565.87   719.2 2563.71
   729.2 2563.64   739.2 2564.79   789.1 2576.28   799.1 2579.91   819.1 2583.45
#Mann= 3 , 0 , 0
       0      .1       0   419.5    .045       0   439.4      .1       0
Bank Sta=419.5,439.4
XS Rating Curve= 0 ,0
Exp/Cntr=0.3,0.1

Type RM Length L Ch R = 1 ,20571   ,315.9,314.2,312.4
XS GIS Cut Line= 3
     1931271.968      249254.661     1931634.968       249444.19
     1931997.968       249633.72
#Sta/Elev= 30
       0 2632.83      20 2621.01    69.9 2601.56    89.9 2595.42   109.9 2588.08
   129.8 2583.44   159.8  2578.1   169.8 2575.22   199.8  2561.6   209.7 2559.14
   249.7 2557.96   269.7 2556.22   319.6 2549.54   339.6 2545.43   349.6 2542.42
   369.6 2536.27   389.5 2528.13   403.5 2526.94   409.5 2526.89   418.5 2526.89
   439.5 2527.37   519.4 2535.73   549.3 2541.67   559.3 2544.68   569.3 2549.48
   579.3 2552.41   589.3 2554.11   649.2 2553.82   659.2 2556.21     819 2582.92
#Mann= 3 , 0 , 0
       0      .1       0   403.5    .045       0   418.5      .1       0
Bank Sta=403.5,418.5
XS Rating Curve= 0 ,0
Exp/Cntr=0.3,0.1

Type RM Length L Ch R = 1 ,20256.8 ,370.3,366.4,362.4
XS GIS Cut Line= 3
     1931124.942      249556.329     1931497.817      249725.157
     1931875.059      249886.336
#Sta/Elev= 30
       0 2583.51    99.8 2568.61   159.7 2571.83   169.7 2571.65   179.7 2569.04
   189.7 2563.77   209.6 2555.51   219.6 2553.45   269.6 2551.89   329.4  2546.5
   349.4 2541.46   359.4 2536.51   369.4  2532.8   389.4 2526.69   399.3  2524.6
   419.3    2523   429.3 2522.69   439.3 2523.18   449.3 2526.27   459.3 2527.98
   519.4 2536.69   539.4  2542.4   549.4 2544.34   569.4 2545.51   609.4 2543.37
   629.4  2543.8   709.5 2550.81   739.5 2554.34   799.5 2563.08   819.6 2566.75
#Mann= 3 , 0 , 0
       0      .1       0   419.3    .045       0   439.3      .1       0
Bank Sta=419.3,439.3
XS Rating Curve= 0 ,0
Exp/Cntr=0.3,0.1

Type RM Length L Ch R = 1 ,19890.4 ,517.3,519.2,520.9
XS GIS Cut Line= 3
      1930962.56      249973.274      1931360.95      250068.014
      1931759.34      250162.754
#Sta/Elev= 30
       0 2609.12      40 2601.75    79.9 2593.04    99.9 2585.82   129.8  2577.9
   169.8 2572.05   189.8 2565.46   229.7 2546.99   239.7 2544.55   289.6 2542.23
   329.6 2539.13   349.6 2536.96   369.6 2533.46   399.5 2526.48   421.6 2520.55
   429.5 2519.63   436.6  2520.1   469.4 2523.54   489.4 2526.36   509.4 2530.44
   549.3 2535.04   559.3 2534.62   599.3 2526.64   609.3 2525.74   619.2 2525.91
   669.2 2535.81   679.2 2539.64   749.1  2554.7   769.1 2560.61     819 2570.26
#Mann= 3 , 0 , 0
       0      .1       0   421.6    .045       0   436.6      .1       0
Bank Sta=421.6,436.6
XS Rating Curve= 0 ,0
Exp/Cntr=0.3,0.1

Type RM Length L Ch R = 1 ,19371.2 ,490.2,486,483.5
XS GIS Cut Line= 3
     1930847.765      250443.643     1931237.091      250570.835
     1931627.326      250694.882
#Sta/Elev= 30
       0 2588.64      40 2583.57      50 2579.85    89.9  2568.9    99.9 2566.56
   119.9 2564.28   129.9  2561.8   139.9 2556.35   169.8 2535.57   179.8 2531.26
   189.8 2529.75   319.7 2525.49   339.6 2521.48   369.6  2512.5   379.6 2510.42
     403 2508.35   409.6 2508.26     418  2508.4   439.5 2509.96   479.5 2518.29
   489.5 2519.12   549.4  2518.1   569.4 2521.54   639.3 2529.61   669.2 2535.26
   719.2 2547.99   749.1 2561.34   779.1 2576.03   809.1 2585.32     819 2589.29
#Mann= 3 , 0 , 0
       0      .1       0     403    .045       0     418      .1       0
Bank Sta=403,418
XS Rating Curve= 0 ,0
Exp/Cntr=0.3,0.1

Type RM Length L Ch R = 1 ,18885.1 ,286.9,287.2,285.8
XS GIS Cut Line= 2
     1930627.341      250909.722     1931442.267      251080.432
#Sta/Elev= 30
       0 2541.86     109 2524.35   118.9 2521.54   188.3 2511.38   208.2 2507.01
   218.1 2506.62     228 2507.37   277.5 2513.37   287.4 2514.11   297.4 2513.68
   327.1  2510.6   356.8 2504.41   366.8 2501.49   405.2 2497.45   416.3 2497.38
   420.2 2497.52   515.4 2504.38   555.1  2508.1     565 2508.14   594.7 2505.83
   614.6 2506.61   664.1 2504.51     674 2506.96   683.9 2513.72   693.8 2525.24
   703.8  2530.3   713.7 2533.75   773.1 2548.12     783 2552.54   832.6 2564.81
#Mann= 3 , 0 , 0
       0      .1       0   405.2    .045       0   420.2      .1       0
Bank Sta=405.2,420.2
XS Rating Curve= 0 ,0
Exp/Cntr=0.3,0.1

Type RM Length L Ch R = 1 ,18597.6 ,380.9,380.8,380.7
XS GIS Cut Line= 2
     1930561.949      251183.695     1931394.003      251325.809
#Sta/Elev= 30
       0 2541.95     9.9 2539.49    29.8 2532.25    89.4 2517.87   109.2  2510.9
   178.8 2494.91   188.7 2494.04   268.1  2502.9     288 2502.64   307.8  2501.2
   327.7 2497.19   347.6 2494.66   417.1 2491.99   466.3 2487.05   466.7 2487.02
   481.3 2487.97   496.5  2490.9   526.3 2493.82     566 2503.17   585.9    2506
   595.8 2505.59   655.4 2497.66   685.2 2497.56   705.1 2500.53     715 2504.33
   724.9  2512.5   744.8 2533.84   764.7 2544.36   834.2 2559.86   844.1 2564.17
#Mann= 3 , 0 , 0
       0      .1       0   466.3    .045       0   481.3      .1       0
Bank Sta=466.3,481.3
XS Rating Curve= 0 ,0
Exp/Cntr=0.3,0.1

Type RM Length L Ch R = 1 ,18216.4 ,560.1,553,545.8
XS GIS Cut Line= 2
     1930414.996      251498.957     1931323.179      251640.973
#Sta/Elev= 30
       0 2562.37      10 2559.46      40 2554.53    79.9 2546.04    89.9 2540.93
   159.9 2520.07   169.9 2515.27   239.8 2495.05   249.8 2491.25   259.8 2489.51
   279.8 2488.86   339.7 2492.96   369.7 2490.04   399.7 2481.09   407.6 2479.69
   409.6 2479.34   422.6 2481.11   429.6 2482.27   489.6 2482.92   549.5 2485.74
   689.4 2496.57   709.4 2495.51   769.4 2487.96   819.3    2489   839.3 2500.11
   859.3 2518.42   869.3  2524.6   899.2 2535.13   909.2 2541.38   919.2 2545.12
#Mann= 3 , 0 , 0
       0      .1       0   407.6    .045       0   422.6      .1       0
Bank Sta=407.6,422.6
XS Rating Curve= 0 ,0
Exp/Cntr=0.3,0.1

Type RM Length L Ch R = 1 ,17663   ,254.3,261.2,268
XS GIS Cut Line= 2
     1930491.833      252165.412     1931312.556      252014.566
#Sta/Elev= 30
       0 2520.68     9.9    2518    19.9  2513.3    29.8 2509.91    89.4 2494.05
   109.3 2486.22     149 2477.57   168.9  2475.8   218.6    2476   248.4 2474.36
   258.3 2472.98     298 2456.64     308 2453.86   317.9 2452.76   425.5 2452.28
   437.1  2451.8   440.5  2451.9   496.7 2455.37   556.3 2460.43   576.2 2463.72
     596 2470.65   615.9 2473.33   665.6 2476.97   705.3 2476.34   715.3 2478.34
   725.2 2482.37     755 2496.58   764.9 2506.43   824.5 2537.65   834.5 2542.26
#Mann= 3 , 0 , 0
       0      .1       0   425.5    .045       0   440.5      .1       0
Bank Sta=425.5,440.5
XS Rating Curve= 0 ,0
Exp/Cntr=0.3,0.1

Type RM Length L Ch R = 1 ,17402.1 ,365.6,362.3,359
XS GIS Cut Line= 2
     1930514.781       252276.76     1931346.197       252393.47
#Sta/Elev= 30
       0    2516      70 2487.28      80 2481.99   119.9 2473.77   129.9 2472.68
   209.9 2470.42   229.9  2467.2   239.9 2463.23   289.8 2451.26   299.8 2450.17
   389.8 2447.16   411.4 2443.55   419.8 2442.37   426.4 2442.83   459.8  2449.3
   549.7  2456.1   559.7 2457.77   579.7 2464.27   599.7 2468.47   609.7  2468.8
   619.7 2467.42   649.7 2459.06   659.7 2457.44   669.6 2458.01   679.6 2459.86
   709.6 2470.02   799.6 2493.68   809.6 2496.76   819.6 2502.03   839.6 2509.75
#Mann= 3 , 0 , 0
       0      .1       0   411.4    .045       0   426.4      .1       0
Bank Sta=411.4,426.4
XS Rating Curve= 0 ,0
Exp/Cntr=0.3,0.1

Type RM Length L Ch R = 1 ,17040   ,434.6,451.7,469.3
XS GIS Cut Line= 2
     1930446.318      252689.909      1931270.75      252684.161
#Sta/Elev= 30
       0 2516.76    59.6 2486.21    69.5 2479.93    79.5 2470.35    99.3 2461.23
   119.2  2460.2   158.9 2463.87   228.5 2462.77   238.4 2457.96   307.9 2436.32
   387.4 2431.98   404.1 2429.34   417.2 2428.68   419.1 2428.79   456.9  2432.6
   526.5 2436.58   546.3 2442.14   556.3 2448.72   566.2 2453.03     596 2460.93
   615.9 2460.47   655.6 2451.27   675.5 2449.97   695.3 2450.64   705.2  2453.5
   715.2 2459.78   725.1 2463.76   784.7 2480.59   804.6 2488.21   824.4 2492.18
#Mann= 3 , 0 , 0
       0      .1       0   404.1    .045       0   419.1      .1       0
Bank Sta=404.1,419.1
XS Rating Curve= 0 ,0
Exp/Cntr=0.3,0.1

Type RM Length L Ch R = 1 ,16588.1 ,373.2,378,382.4
XS GIS Cut Line= 3
     1930380.163      252805.706     1930688.048      253076.534
     1930982.404      253361.078
#Sta/Elev= 30
       0 2520.97      60 2475.79      80 2458.64      90  2453.9     100 2451.91
     200 2455.97     230 2447.74     280 2431.27     300 2423.08     310 2420.58
     360 2409.79   412.7  2402.8     420 2402.36   427.7 2402.99     440 2406.73
     460 2416.08   499.9 2420.73   509.9 2423.96   539.9 2439.54   549.8 2442.76
   559.8 2443.91   569.8 2442.92   619.7 2434.27   639.7  2429.5   669.7  2426.6
   679.7 2427.83   699.6 2436.13   739.6 2443.99   759.5 2451.21   819.4 2465.52
#Mann= 3 , 0 , 0
       0      .1       0   412.7    .045       0   427.7      .1       0
Bank Sta=412.7,427.7
XS Rating Curve= 0 ,0
Exp/Cntr=0.3,0.1

Type RM Length L Ch R = 1 ,16210.1 ,427.9,438.8,449.7
XS GIS Cut Line= 3
     1930176.663      252995.639     1930411.788       253330.91
     1930646.913       253666.18
#Sta/Elev= 30
       0 2566.04      20 2558.35      30 2549.68    49.9 2520.77    59.9 2517.04
   119.8 2446.31   129.8 2438.63   139.8 2436.66   149.8 2437.43   259.7 2452.54
   269.7 2452.73   299.6  2443.8   379.5 2399.29   389.5 2395.02   404.7  2392.1
   419.5 2391.42   419.7 2391.42   429.5 2391.66   459.4 2400.17   499.4 2404.04
   529.4 2412.42   559.3 2425.58   579.3 2432.05   589.3 2432.94   599.3 2431.66
   679.2 2418.29   719.1 2416.89   729.1 2417.64   749.1 2428.19     819 2441.36
#Mann= 3 , 0 , 0
       0      .1       0   404.7    .045       0   419.7      .1       0
Bank Sta=404.7,419.7
XS Rating Curve= 0 ,0
Exp/Cntr=0.3,0.1

Type RM Length L Ch R = 1 ,15771.2 ,368.8,361.6,354.5
XS GIS Cut Line= 2
     1929968.704      253107.146     1930074.919      253919.712
#Sta/Elev= 30
       0 2535.22      20 2529.02      30 2528.82      70 2512.42      80 2506.14
   119.9  2467.8   129.9 2467.18   169.9 2427.83   179.9 2422.81   229.8 2424.06
   259.8 2420.03   269.8 2417.01   299.8  2398.3   309.8 2396.91   329.8 2390.03
   369.8 2381.54   408.1 2378.36   419.7 2378.06   423.1 2378.47   449.7 2383.84
   539.7 2388.61   569.6 2396.93   589.6 2405.96   619.6  2416.1   629.6    2418
   719.5 2412.82   729.5 2414.43   769.5 2425.93   789.5 2428.42   819.5 2437.12
#Mann= 3 , 0 , 0
       0      .1       0   408.1    .045       0   423.1      .1       0
Bank Sta=408.1,423.1
XS Rating Curve= 0 ,0
Exp/Cntr=0.3,0.1

Type RM Length L Ch R = 1 ,15409.6 ,419.5,420,420.5
XS GIS Cut Line= 3
     1929503.881      253256.644     1929680.782      253625.962
     1929857.683      253995.281
#Sta/Elev= 30
       0 2457.53    49.9 2445.92    79.9  2442.5   119.8 2433.44   159.8 2420.08
   179.8 2416.45   209.7 2406.15   229.7 2400.87   299.6  2403.9   339.6 2399.15
   349.6 2395.25   379.5 2380.01   389.5 2377.98   399.5 2371.23   404.9 2369.36
   409.5 2367.76   419.9 2368.34   449.4 2374.11   509.4 2378.11   539.3 2382.42
   569.3 2391.16   589.3 2394.44   629.2 2406.56   649.2 2408.15   699.2 2407.28
   709.1  2409.2     779 2438.36     789 2441.68     799 2442.41     819 2450.54
#Mann= 3 , 0 , 0
       0      .1       0   404.9    .045       0   419.9      .1       0
Bank Sta=404.9,419.9
XS Rating Curve= 0 ,0
Exp/Cntr=0.3,0.1

Type RM Length L Ch R = 1 ,14989.6 ,386.9,379.1,371.3
XS GIS Cut Line= 3
     1929132.412      253432.246     1929301.272      253805.309
     1929470.133      254178.373
#Sta/Elev= 30
       0 2418.62    69.9 2403.28    79.9 2403.21   129.8 2393.12   169.8 2386.24
   179.8 2386.27   219.7 2378.91   239.7 2377.94   299.6  2381.4   339.6 2378.18
   349.6 2376.44   379.5  2367.2   389.5  2366.6   408.2    2359   419.5 2356.58
   423.2 2357.18   459.4 2366.98   489.4 2370.34   539.3 2379.05   589.3 2394.04
   629.2 2395.67   659.2 2393.34   669.2  2394.2   699.2 2405.54   709.1 2415.84
   719.1 2424.18   729.1 2430.15     779 2456.94     799 2462.76     819 2474.93
#Mann= 3 , 0 , 0
       0      .1       0   408.2    .045       0   423.2      .1       0
Bank Sta=408.2,423.2
XS Rating Curve= 0 ,0
Exp/Cntr=0.3,0.1

Type RM Length L Ch R = 1 ,14610.5 ,399.3,400,400.6
XS GIS Cut Line= 3
     1928698.532      253714.985      1928982.74      254009.806
     1929268.072      254303.533
#Sta/Elev= 30
       0 2383.85    69.9  2370.8   149.8 2362.96   259.7 2367.31   279.7 2366.11
   319.6 2359.47   369.6 2360.91   379.5 2359.44   404.3  2348.2   409.5 2346.22
   419.3  2347.5   439.5 2359.96   459.4  2368.8   469.4 2371.91   489.4 2374.98
   529.4 2383.91   539.3 2385.47   589.3 2386.44   629.2 2383.75   639.2 2386.73
   659.2 2407.18   689.2 2433.38   709.1 2453.95   719.1  2463.1   729.1 2468.92
   739.1 2470.39   759.1 2477.76     789 2486.32     799 2488.09     819 2488.64
#Mann= 3 , 0 , 0
       0     .06       0   404.3    .045       0   419.3     .06       0
Bank Sta=404.3,419.3
XS Rating Curve= 0 ,0
Exp/Cntr=0.3,0.1

Type RM Length L Ch R = 1 ,14210.4 ,449.2,449.1,449.2
XS GIS Cut Line= 3
     1928407.417       253968.63     1928681.893      254272.516
     1928960.407      254572.776
#Sta/Elev= 30
       0 2370.33      40 2361.24    79.9 2355.69   119.8 2357.61   149.8 2362.25
   169.8 2362.25   179.8 2360.79   209.7 2350.58   249.7 2347.47   269.7 2348.92
   289.6 2357.52   299.6 2359.96   349.6 2358.83   369.5 2354.98   404.4 2338.45
   409.5 2336.19   419.4 2334.79   429.5 2336.01   479.4 2354.95   499.4 2359.69
   519.4 2369.67   529.4 2373.06   549.3 2374.62   589.3 2370.61   599.3 2371.52
   629.2 2381.76   699.2 2395.11   749.1 2407.41   759.1 2408.85     819  2426.1
#Mann= 3 , 0 , 0
       0     .06       0   404.4    .045       0   419.4     .06       0
Bank Sta=404.4,419.4
XS Rating Curve= 0 ,0
Exp/Cntr=0.3,0.1

Type RM Length L Ch R = 1 ,13761.4 ,340.3,352.1,362
XS GIS Cut Line= 3
     1928064.615      254263.849     1928342.561      254564.575
     1928619.881       254865.88
#Sta/Elev= 30
       0 2363.38      10 2357.17      20 2354.07      30 2354.82    49.9 2359.98
    59.9 2360.44   139.8 2355.12   179.8 2353.53   209.7 2350.78   219.7 2351.58
   239.7 2348.25   289.6 2334.38   369.6 2332.45   399.5 2326.56   408.7  2326.6
   423.7 2329.14   519.4 2348.57   529.4 2351.59   549.3 2360.98   569.3  2365.6
   589.3 2366.39   609.3 2365.51   659.2  2354.4   669.2 2356.74   719.1 2374.55
   729.1 2377.34   739.1 2378.57   759.1 2385.31     779 2393.85     819 2407.47
#Mann= 3 , 0 , 0
       0      .1       0   408.7    .045       0   423.7      .1       0
Bank Sta=408.7,423.7
XS Rating Curve= 0 ,0
Exp/Cntr=0.3,0.1

Type RM Length L Ch R = 1 ,13409.3 ,417.3,398.7,382.4
XS GIS Cut Line= 3
     1927967.031      254333.939     1928063.335      254752.488
     1928193.955      255148.379
#Sta/Elev= 30
       0 2355.72      10 2354.15      40  2358.8    59.9 2357.69    69.9 2356.42
    99.9 2349.53   119.9 2339.96   129.8 2336.14   139.8 2334.02   199.8 2329.21
   269.7 2320.17   359.6  2315.6   379.6 2315.02     489 2317.38   518.8 2320.18
   558.5 2325.46   578.4 2326.85   608.2 2331.59   637.9  2340.2   667.7 2347.15
   677.6  2348.5   697.5  2357.7   707.4  2360.4   727.3 2360.66     757 2358.92
     767 2358.92   776.9 2360.21   786.8 2363.93   806.7 2373.57   846.4 2398.84
#Mann= 3 , 0 , 0
       0      .1       0   359.6    .045       0   379.6      .1       0
Bank Sta=359.6,379.6
XS Rating Curve= 0 ,0
Exp/Cntr=0.3,0.1

Type RM Length L Ch R = 1 ,13010.2 ,273.6,285.1,296.1
XS GIS Cut Line= 3
     1927430.136      254747.656     1927781.928      254960.333
      1928110.52      255212.831
#Sta/Elev= 30
       0 2352.38     9.8 2349.43    19.6 2345.86    39.2  2336.9    58.7 2330.52
    88.1 2326.84     137 2324.14   303.4 2317.02   342.6  2314.7   362.1 2312.42
   384.8 2308.27   391.5 2307.02   399.8 2306.73   401.3 2306.68     421 2314.31
   430.8 2316.44   509.8 2325.84   578.8 2340.04   588.7 2341.84   608.4 2343.76
   628.2 2348.05   647.9 2351.29   687.4 2356.62     717 2359.42   736.7 2359.56
   756.4 2358.77   766.3 2359.64   776.2 2365.05   805.8  2386.4   825.5 2398.83
#Mann= 3 , 0 , 0
       0      .1       0   384.8    .045       0   399.8      .1       0
Bank Sta=384.8,399.8
XS Rating Curve= 0 ,0
Exp/Cntr=0.3,0.1

Type RM Length L Ch R = 1 ,12725.1 ,429,416.2,403.3
XS GIS Cut Line= 2
     1927373.011      254815.627     1927758.998      255486.677
#Sta/Elev= 30
       0 2343.79     9.9 2336.45    19.8 2330.14    29.8 2326.92   168.7 2316.66
   188.6    2316     258 2311.87   297.8 2311.24   317.6 2310.32   367.2 2302.03
     374 2301.57   377.2 2301.35     389 2302.61     397 2304.06   406.9 2304.89
   426.8 2309.65   446.6 2313.17   535.9  2322.3   555.8 2325.27   575.6  2331.5
   595.5 2339.62   605.4 2343.01   615.3 2344.92     665 2365.04   674.9 2367.53
   684.8 2366.47   714.6  2359.5   734.4 2356.84   744.4 2355.59   774.1 2355.06
#Mann= 3 , 0 , 0
       0      .1       0     374    .045       0     389      .1       0
Bank Sta=374,389
XS Rating Curve= 0 ,0
Exp/Cntr=0.3,0.1

Type RM Length L Ch R = 1 ,12308.8 ,483.5,518.1,546.5
XS GIS Cut Line= 2
     1926919.742      255233.484     1927912.542      255766.986
#Sta/Elev= 30
       0 2346.07    49.9 2345.11   129.7 2337.42   139.6 2333.88   149.6 2327.92
   159.6 2316.94   169.6 2311.78   179.5 2309.64   309.2 2308.68     369 2297.66
   377.7 2297.21     379 2297.14   392.7 2298.21   448.8 2305.69   528.6 2310.62
   598.4 2317.24   658.3 2328.64   718.1  2349.2     778 2354.56   817.9  2354.3
   827.8 2355.79   837.8 2359.69   877.7 2384.96   887.7 2393.36   897.7    2404
   907.6 2405.74   937.6 2405.49   977.4 2408.91   997.4 2412.54  1127.1 2428.57
#Mann= 3 , 0 , 0
       0      .1       0   377.7    .045       0   392.7      .1       0
Bank Sta=377.7,392.7
XS Rating Curve= 0 ,0
Exp/Cntr=0.3,0.1

Type RM Length L Ch R = 1 ,11790.6 ,294.5,284.7,274.9
XS GIS Cut Line= 3
     1926856.408      255187.954     1926909.118      255422.936
     1926896.525      256272.362
#Sta/Elev= 30
       0 2351.86    28.9 2345.54   154.1 2344.01   240.8 2336.63   310.8 2333.94
   320.8 2331.96   330.8 2326.56   350.8 2318.06   360.8 2309.69   370.8 2303.76
   380.7 2299.87   410.7 2292.07   423.2 2289.89   438.2 2289.35   440.7 2289.34
   450.7 2290.71   490.7 2304.29   570.6 2312.58   620.6 2319.28   640.6 2320.78
   710.6 2332.71   730.5 2334.71   810.5 2355.06   850.5 2361.22   880.5 2363.04
   940.4 2363.19   980.4 2361.56  1010.4 2361.79  1040.4 2357.78  1090.3 2360.06
#Mann= 3 , 0 , 0
       0      .1       0   423.2    .045       0   438.2      .1       0
Bank Sta=423.2,438.2
XS Rating Curve= 0 ,0
Exp/Cntr=0.3,0.1

Type RM Length L Ch R = 1 ,11505.9 ,664.9,665.3,665.6
XS GIS Cut Line= 3
     1926480.175      255277.914     1926742.684      255909.846
     1926786.619      256045.908
#Sta/Elev= 30
       0  2345.1    19.8 2344.44    49.6 2341.18    79.3  2341.1   109.1 2342.79
   178.5 2349.24   198.3 2349.32     238 2347.26   247.9 2345.21   257.8 2341.51
   267.8 2340.77   277.7 2337.16   317.4 2315.35   347.1 2303.76     357 2300.52
   366.9  2299.9   396.7    2291   406.6 2289.35   416.5 2289.65   466.1 2300.11
     476 2300.38   575.2  2318.7   585.1 2319.18   664.4 2335.85   693.8 2339.92
   722.4 2342.31   760.5 2353.67   779.6 2357.78   789.1 2358.33   827.3 2367.74
#Mann= 3 , 0 , 0
       0      .1       0   396.7    .045       0   416.5      .1       0
Bank Sta=396.7,416.5
XS Rating Curve= 0 ,0
Exp/Cntr=0.3,0.1

Type RM Length L Ch R = 1 ,10840.4 ,395.4,373,350.6
XS GIS Cut Line= 2
      1925942.38      255242.337     1926234.526      256021.393
#Sta/Elev= 30
       0 2399.87    59.4 2391.51      99  2384.7   138.7 2374.82   168.4 2365.67
   188.2  2360.6   198.1 2359.83   247.6 2341.72   257.5 2340.18   326.9 2339.65
   356.6 2337.07   366.5  2335.4   376.4  2331.1   386.3 2328.67   396.2 2324.29
     416 2309.85   445.7 2290.75   455.6 2289.18   474.7  2290.2   495.3 2296.95
   505.2 2297.89   594.3 2312.78   604.2 2312.74   614.1 2314.34   683.5 2329.35
   703.3 2330.97   762.7 2343.24   792.4 2351.72   812.2 2355.26     832 2361.84
#Mann= 3 , 0 , 0
       0      .1       0   455.6    .045       0   474.7      .1       0
Bank Sta=455.6,474.7
XS Rating Curve= 0 ,0
Exp/Cntr=0.3,0.1

Type RM Length L Ch R = 1 ,10467.2 ,317.3,310,302.5
XS GIS Cut Line= 2
     1925342.153      255865.582     1926393.879      256109.922
#Sta/Elev= 30
       0 2373.35      60 2373.04      80 2370.85     100  2356.4     130 2346.29
     160 2342.56     210 2342.41   229.9 2344.61   249.9 2353.87   269.9 2366.77
   279.9 2369.96   339.9  2368.9   369.9 2362.51   439.9 2339.24   509.9 2325.69
   539.9 2314.87   579.9  2293.8   589.9 2290.13   599.8 2289.23   610.6  2289.3
   625.6 2289.78   649.8 2294.39   669.8 2305.59   689.8 2319.66   769.8 2331.53
   849.8 2353.26   859.8 2358.84   889.8 2365.66   959.8  2374.2  1079.7 2372.84
#Mann= 3 , 0 , 0
       0      .1       0   610.6    .045       0   625.6      .1       0
Bank Sta=610.6,625.6
XS Rating Curve= 0 ,0
Exp/Cntr=0.3,0.1

Type RM Length L Ch R = 1 ,10157.1 ,320.1,321.1,322.3
XS GIS Cut Line= 3
     1925703.352      256311.768     1925855.622      256313.539
     1926344.303      256253.339
#Sta/Elev= 30
       0 2365.31    66.6 2366.77   104.7 2366.76   114.2 2365.97   123.7 2363.63
   133.2  2359.8   142.8 2352.13   152.3 2345.59   211.4 2315.46   231.1 2304.43
   260.6 2293.21   270.4  2290.1   280.3 2289.13   290.9 2289.41     300 2290.54
   305.9 2292.34   309.8 2293.53   349.2 2300.62   359.1  2300.9   388.6 2308.27
   398.5 2313.55   467.4 2333.19   477.2 2338.36   487.1 2341.76   536.3 2355.93
     556 2360.57   575.7 2366.36   595.4 2369.54     625 2372.51   644.7 2376.08
#Mann= 3 , 0 , 0
       0      .1       0   290.9    .045       0   305.9      .1       0
Bank Sta=290.9,305.9
XS Rating Curve= 0 ,0
Exp/Cntr=0.3,0.1

Type RM Length L Ch R = 1 ,9835.8  ,361.5,389.4,417.3
XS GIS Cut Line= 3
     1925844.998      256610.997     1925937.069      256605.685
     1926466.602      256570.029
#Sta/Elev= 30
       0 2335.34    18.4 2337.09    36.9 2337.47      83 2336.16    92.2 2334.94
     102  2332.9     161 2317.84   180.7 2310.29   200.3 2305.69     220 2303.61
   249.5 2297.17   266.9 2290.97   269.1 2290.12     279  2289.2   281.9 2289.38
   288.8  2289.8   298.6  2292.3   328.1 2305.01   337.9 2309.81   347.8 2317.01
   416.6  2344.5   426.4 2351.97   455.9 2362.87   465.7 2365.49   495.2  2369.6
     505 2371.86   573.8 2380.58   583.6 2382.35   593.5 2382.93     623 2380.95
#Mann= 3 , 0 , 0
       0      .1       0   266.9    .045       0   281.9      .1       0
Bank Sta=266.9,281.9
XS Rating Curve= 0 ,0
Exp/Cntr=0.3,0.1

Type RM Length L Ch R = 1 ,9446.7  ,516.7,542.1,567.4
XS GIS Cut Line= 3
     1925883.951      256644.638     1925906.969      256722.543
      1926124.75      257250.177
#Sta/Elev= 30
       0 2332.83       9 2331.84    36.1 2325.82    54.2 2322.69    63.2 2322.11
   100.9 2322.32     160 2319.53   199.3 2314.71   258.4 2299.57   287.9 2290.92
   297.8 2289.26   307.6 2289.21   308.7 2289.25   317.4 2289.58   323.7 2291.36
   327.3 2292.37   337.1 2296.82   376.5 2312.43   386.3 2315.96     406 2319.79
   455.2 2338.95   484.7 2349.26   494.6 2353.72   514.3 2358.94     534 2368.04
   543.8 2370.72   553.6 2371.22   612.7 2371.62   642.2 2371.67     652 2371.29
#Mann= 3 , 0 , 0
       0      .1       0   308.7    .045       0   323.7      .1       0
Bank Sta=308.7,323.7
XS Rating Curve= 0 ,0
Exp/Cntr=0.3,0.1

Type RM Length L Ch R = 1 ,8904.3  ,523.8,496.1,468.3
XS GIS Cut Line= 3
     1925800.658      256459.522     1925482.029      256821.696
     1925478.488      257147.483
#Sta/Elev= 30
       0 2350.86    88.6 2343.98   108.3 2338.66   118.1 2336.87   167.4 2314.79
     187 2303.51   216.6 2291.92   226.4  2289.4   246.1 2289.06   248.8 2289.28
   263.8 2291.28   285.5 2294.91   295.3 2297.69   305.2 2301.72   334.7 2309.32
   354.4 2313.63   374.1 2315.08   413.5 2322.41   462.7 2329.76   492.3 2331.53
   571.2 2341.26   581.1 2341.45   650.2 2351.75   660.1 2352.95     670 2352.96
   689.7 2355.38   758.8 2366.43   768.7 2366.63   778.6 2368.08   808.2 2373.68
#Mann= 3 , 0 , 0
       0      .1       0   248.8    .045       0   263.8      .1       0
Bank Sta=248.8,263.8
XS Rating Curve= 0 ,0
Exp/Cntr=0.3,0.1

Type RM Length L Ch R = 1 ,8408.3  ,208.9,208.1,207.4
XS GIS Cut Line= 4
     1924901.202      256001.531     1924999.415      256286.657
     1925374.024      256961.572     1925381.458      257139.735
#Sta/Elev= 30
       0 2418.65    97.3 2418.13   145.9 2415.47   252.9 2387.01   272.4 2384.05
   301.6  2375.7   331.2 2365.37   370.8 2345.99   380.7 2342.46   400.5 2339.46
   469.8 2337.24   509.4 2339.13   519.3 2336.73     549 2325.62   578.7    2312
   588.6 2310.91     638 2291.75   647.9 2289.95   687.5    2289   707.3    2289
   717.2 2290.05   727.1 2295.13     737 2298.36   875.6 2316.67   905.2 2322.02
  1073.5 2346.34  1132.9 2352.39  1212.2 2364.63  1222.1 2364.78  1251.8 2370.89
#Mann= 3 , 0 , 0
       0      .1       0   687.5    .045       0   707.3      .1       0
Bank Sta=687.5,707.3
XS Rating Curve= 0 ,0
Exp/Cntr=0.3,0.1

Type RM Length L Ch R = 1 ,8200.2  ,549.3,533,516.7
XS GIS Cut Line= 2
     1924816.096      256422.635     1925286.163      257180.995
#Sta/Elev= 30
       0 2367.21    19.8 2362.22    29.7 2361.53    99.1  2345.6     119 2340.03
   158.6 2334.09   188.4    2332   247.8 2330.37   267.7 2328.26   317.2 2321.09
   327.2 2317.95     347 2307.25   356.9 2304.54   390.7 2291.31   396.6 2289.55
   405.7 2288.95   406.5  2288.9   416.4 2291.36   436.2 2297.86     456 2300.88
   465.9 2301.21   525.4 2310.95   703.9 2330.83   733.6 2336.31   753.4 2344.06
   763.4  2347.4   773.3 2349.58   783.2 2351.58     803 2353.77   892.2 2370.16
#Mann= 3 , 0 , 0
       0      .1       0   390.7    .045       0   405.7      .1       0
Bank Sta=390.7,405.7
XS Rating Curve= 0 ,0
Exp/Cntr=0.3,0.1
